HEC-RAS study BOGGSCK.prj: BOGGSCK

--- BOGGSCK.g01 (geometry) --- (continued)

Type RM Length L Ch R = 1 ,18022   ,458.5,526.3,295.9
XS GIS Cut Line= 5
     2036800.411      337485.415     2037119.034      337603.707
     2037188.674       337715.32     2037283.116      337802.131
2037616.21161213337941.896356288
#Sta/Elev= 30
       0 2468.15    2.112467.997   91.152462.506   146.5 2460.41   163.7 2456.69
  171.842453.112     178 2450.52     185 2449.32  217.182448.475   352.2 2449.47
     360 2445.66   375.4 2443.53   383.22445.887     387 2447.27   402.5 2446.79
     418 2448.82   437.3 2449.44   463.6 2448.16   518.3 2449.14   568.3 2448.27
   593.8 2450.39   616.6 2450.48   655.7 2448.82   684.2 2451.45   726.9 2457.11
   768.8 2457.42     798 2461.89   845.1 2464.06   922.6 2473.87   960.9 2477.14
#Mann= 7 ,-1 , 0
       0     .12       0    2.11     .06       0   91.15     .12       0
  171.84    .016       0  217.18     .12       0     360    .045       0
   383.2     .12       0
#XS Ineff= 2 , 0
             226    2460
Permanent Ineff=
       F       F
Bank Sta=360,383.2
XS Rating Curve= 0 ,0
Exp/Cntr=0.3,0.1

Type RM Length L Ch R = 1 ,17495.7 ,326.2,291.9,337.6
XS GIS Cut Line= 4
     2036855.408      337730.567     2036985.147       337846.95
     2037040.477      337920.4052037377.28931365338281.075929883
#Sta/Elev= 30
       0 2462.01   32.072461.507    59.6  2460.2   76.312454.336    87.4 2449.56
      93 2448.42   115.3 2448.43   145.9 2445.65   159.8 2446.08   175.7    2448
   189.8 2447.82   196.92444.715   199.2 2443.69   210.1  2442.7   219.7 2444.76
   240.2 2447.52   264.8 2449.16   329.8 2448.05   341.7 2449.18  442.122448.784
   561.9 2449.25     588 2453.49  597.692459.896   617.6 2467.88   631.5 2471.91
   673.3 2479.41   691.2 2480.51   713.7 2484.57   731.4 2489.11   759.7 2498.38
#Mann= 7 ,-1 , 0
       0     .12       0   32.07    .016       0   76.31     .12       0
   196.9    .045       0   219.7     .12       0  442.12     .08       0
  597.69     .12       0
Bank Sta=196.9,219.7
XS Rating Curve= 0 ,0
Exp/Cntr=0.3,0.1

Type RM Length L Ch R = 1 ,17203.8 ,361.9,504.3,444.2
XS GIS Cut Line= 4
     2036713.268      337893.694      2036761.92       337998.63
     2036856.362      338162.7122037134.98331365338507.075247634
#Sta/Elev= 30
       0 2457.58    6.582457.287    31.9 2457.16    39.1 2456.06    49.9 2447.87
    53.6 2446.97   126.3 2447.69   130.1 2447.23   135.9  2443.7   145.5 2442.38
   157.82443.525   164.2 2447.73     168 2448.28   202.1  2444.6   232.4 2447.55
     274 2444.83   285.4 2448.08   292.9 2447.37   322.8 2448.59   366.6 2446.68
  440.262447.256  504.062448.994   527.9 2449.97   539.7 2452.72   553.2  2453.3
   561.6 2456.23   637.9 2469.59     646 2472.78   691.4 2484.03   747.9 2505.77
#Mann= 6 ,-1 , 0
       0     .06       0    6.58     .12       0   135.9    .045       0
   157.8     .12       0  440.26     .08       0  504.06     .12       0
Bank Sta=135.9,157.8
XS Rating Curve= 0 ,0
Exp/Cntr=0.3,0.1

Type RM Length L Ch R = 1 ,16699.6 ,286.6,362.5,331.4
XS GIS Cut Line= 4
     2036439.481      338073.993     2036672.248      338197.054
     2036750.473      338213.2722037078.72716235338590.835266902
#Sta/Elev= 30
       0    2465    6.192462.585    21.8 2461.27    33.3 2457.28    58.9 2453.33
   69.392447.241    81.2  2445.6   103.5  2447.7   207.4  2447.9   249.4 2446.51
   269.6 2447.78   286.5 2446.99   292.42443.796   296.6 2442.05     310 2441.96
   316.5 2443.75   326.7  2446.3   353.5 2448.06   388.5 2447.09   401.5 2448.62
   451.3 2449.05     549 2452.87   607.1  2453.5   618.7 2452.28   648.7 2456.45
   690.8 2459.12   711.8 2464.91   733.7 2468.69   757.9 2476.32   843.5 2497.52
#Mann= 5 ,-1 , 0
       0     .12       0    6.19    .016       0   69.39     .12       0
   292.4    .045       0   316.5     .12       0
Bank Sta=292.4,316.5
XS Rating Curve= 0 ,0
Exp/Cntr=0.3,0.1

Type RM Length L Ch R = 1 ,16337.1 ,355,419.6,334.4
XS GIS Cut Line= 4
     2036370.796      338165.574     2036501.488      338308.668
     2036521.522      338410.7422036760.90416646338751.073418196
#Sta/Elev= 30
       0 2457.71     8.8  2456.1      32 2456.16    39.92454.421      83 2447.57
   119.7 2448.29   146.4 2444.74   201.6 2446.81   208.3  2446.5  211.312443.571
   228.2 2441.72   241.7 2442.23   244.22443.954   251.7 2447.09   275.7 2444.84
   288.5 2446.54   348.4 2446.89     399 2444.86   445.4  2445.7     477 2444.57
   491.1 2449.03   507.3 2450.93   518.7 2455.51   576.5 2466.94   627.6  2474.6
   639.6 2474.79   671.7 2484.45   681.9 2485.54     702 2493.44   713.9 2496.46
#Mann= 4 ,-1 , 0
       0    .016       0    39.9     .12       0  211.31    .045       0
   244.2     .12       0
Bank Sta=211.31,244.2
XS Rating Curve= 0 ,0
Exp/Cntr=0.3,0.1

Type RM Length L Ch R = 1 ,15917.5 ,366.1,395.5,426.8
XS GIS Cut Line= 3
     2036142.269       338417.42     2036287.483      338508.576
     2036543.993      338690.889
#Sta/Elev= 30
       0 2513.06    21.2 2498.52   40.952489.353    52.2 2482.26      61 2474.55
    71.6 2471.77   81.722465.536    87.1  2462.1    96.7 2453.03   102.5 2450.74
     111 2449.56   122.9 2443.12   129.7 2441.13   145.2  2441.4   149.2 2443.04
   152.9 2445.77   156.8 2446.72     185 2442.58   216.6    2443   248.2  2445.1
   264.6 2443.15   281.3 2443.29   292.6 2445.76   325.3  2444.2   358.8  2445.9
   371.9 2449.47   389.7 2449.54   401.1 2455.57   415.2 2458.56   486.2 2467.37
#Mann= 5 ,-1 , 0
       0     .12       0   40.95    .016       0   81.72     .12       0
   122.9    .045       0   149.2     .12       0
Bank Sta=122.9,149.2
XS Rating Curve= 0 ,0
Exp/Cntr=0.3,0.1

Type RM Length L Ch R = 1 ,15522   ,312.1,363.2,383.6
XS GIS Cut Line= 4
     2036038.333      338668.959     2036121.997      338732.835
      2036149.55      338805.226     2036288.302        338909.5
#Sta/Elev= 30
       0 2486.88    17.1 2479.27    36.7 2468.86    41.9 2465.53   46.482464.262
    54.3 2462.94    62.5 2459.54    66.7 2457.08    70.8 2453.39    74.9 2450.58
   95.152446.945   108.9 2444.94   119.7 2442.58   126.5 2441.06     144 2440.83
   147.5 2441.03     151  2442.8   154.5 2445.61   158.1 2445.91   175.5 2445.58
     209 2446.74   264.5 2445.35   290.5 2445.73   302.7 2448.81   312.1 2448.78
   315.1 2449.85   323.3 2455.13   333.2 2458.89   343.8 2462.28   356.3 2465.01
#Mann= 5 ,-1 , 0
       0     .12       0   46.48    .016       0   95.15     .12       0
   119.7    .045       0     151     .12       0
Bank Sta=119.7,151
XS Rating Curve= 0 ,0
Exp/Cntr=0.3,0.1

Type RM Length L Ch R = 1 ,15158.7 ,282.2,264.3,240
XS GIS Cut Line= 4
     2035866.546      338839.576      2036023.95      339011.289
     2036034.443      339106.685     2036106.945      339183.956
#Sta/Elev= 30
       0 2485.36    37.2 2469.23   47.222465.859    64.6 2461.12      72 2457.92
    82.4 2456.91   87.292455.365    94.7  2451.5    99.6  2449.9     119 2446.75
   157.9 2445.03   182.1 2444.92   229.2 2446.91   240.1 2445.51     250  2445.4
   263.42442.411   269.8 2441.06   289.6 2440.85   294.5 2442.75   306.1 2445.35
   315.3 2445.87   325.9 2448.09   342.8 2449.88   348.5 2452.11   359.3 2458.57
   378.5 2464.72   387.9 2468.53   396.8 2470.79   406.5 2475.82   434.9 2486.14
#Mann= 5 ,-1 , 0
       0     .12       0   47.22    .016       0   87.29     .12       0
   263.4    .045       0   294.5     .12       0
Bank Sta=263.4,294.5
XS Rating Curve= 0 ,0
Exp/Cntr=0.3,0.1

Type RM Length L Ch R = 1 ,14894.4 ,285,297.6,305.7
XS GIS Cut Line= 4
     2035667.092      338924.818     2035779.447      339130.429
     2035820.756      339197.312     2035878.981      339282.861
#Sta/Elev= 30
       0 2475.44     8.9  2470.5    22.6 2465.77    36.3 2463.26    54.3 2462.46
   77.162458.229    96.3 2454.25  110.822446.493   114.1 2445.31   117.9 2444.91
   138.9  2444.1     180 2446.25   200.3 2445.75   207.6 2444.93   241.3 2445.96
   249.2 2445.55     2542442.694   257.9 2440.55   265.1 2440.34     280 2441.38
   284.6 2442.64   293.7  2445.6   318.7 2447.67   326.7 2449.87   344.8 2458.85
   354.5 2460.88   362.3  2466.8   378.9 2474.13   398.1 2485.06   416.4 2493.27
#Mann= 5 ,-1 , 0
       0     .12       0   77.16    .016       0  110.82     .12       0
     254    .045       0   284.6     .12       0
Bank Sta=254,284.6
XS Rating Curve= 0 ,0
Exp/Cntr=0.3,0.1

Type RM Length L Ch R = 1 ,14596.8 ,318.1,411,389
XS GIS Cut Line= 4
     2035461.845      339035.159     2035517.493      339168.258
     2035538.383       339245.01     2035643.601      339411.274
#Sta/Elev= 30
       0 2496.68     6.9 2495.89      42 2479.95   49.842477.512    63.6 2469.88
    74.3 2467.23    81.4 2463.38   92.662462.001   106.3 2456.33   117.2 2447.63
   120.5 2446.58   127.6 2446.01   139.8 2443.27   162.4 2444.56   165.8 2444.38
  170.22 2442.39     176 2440.24   196.4 2441.17  200.52 2442.57   203.2 2445.05
   206.6 2445.81   223.6 2445.63   235.2 2444.43   265.3 2445.58   294.6 2445.16
   315.3 2442.89   346.2 2444.84   358.1 2447.72   411.2 2468.12   420.6 2469.39
#Mann= 5 ,-1 , 0
       0     .12       0   49.84    .016       0   92.66     .12       0
  170.22    .045       0  200.52     .12       0
Bank Sta=170.22,200.52
XS Rating Curve= 0 ,0
Exp/Cntr=0.3,0.1

Type RM Length L Ch R = 1 ,14185.8 ,289.5,228.3,166.4
XS GIS Cut Line= 3
     2035239.899      339231.654     2035321.516      339393.828
     2035437.051      339517.843
#Sta/Elev= 30
       0 2482.25    14.7 2477.92    36.7 2469.22    40.4 2466.88    45.2 2462.33
   47.582460.763    55.1  2459.7    58.8 2457.89    66.1 2450.08    76.7 2441.32
    80.8 2440.29    84.5 2440.18      99 2440.25   102.8 2440.57   104.72441.386
   110.2 2444.62  113.28 2445.02   125.9 2445.75   149.7 2443.64   157.9  2443.4
  162.17 2443.94     169 2445.11  178.982444.352   198.3 2443.58   228.5 2446.86
   256.3  2447.6   266.4 2448.55   314.4 2450.28   337.6 2451.67     351 2451.79
#Mann= 7 ,-1 , 0
       0     .12       0   47.58    .016       0    76.7    .045       0
   104.7    .016       0  113.28     .12       0  162.17    .016       0
  178.98     .12       0
Bank Sta=76.7,104.7
XS Rating Curve= 0 ,0
Exp/Cntr=0.3,0.1

Type RM Length L Ch R = 1 ,13957.5 ,149.9,127.4,106.7
XS GIS Cut Line= 3
     2035075.605      339527.382     2035319.425      339522.271
     2035415.841      339525.102
#Sta/Elev= 30
       0 2469.74    15.1 2465.58    44.6 2459.48    54.4    2456    70.9 2447.38
    74.1 2446.41    77.4 2446.09    87.3 2446.33   110.2 2444.82   123.4 2445.16
   135.6 2444.09   146.3 2444.59   149.6 2444.36  154.06 2441.92   156.2 2440.68
   159.5 2440.07   182.4 2440.12   185.7 2440.54     189 2441.95   192.3 2443.51
   195.2 2444.17   208.7 2445.29   215.2 2447.12   218.5 2447.43   225.1 2446.25
   231.7 2445.83   244.8 2447.41     262  2447.1  274.362447.904   340.3 2451.45
#Mann= 4 ,-1 , 0
       0     .12       0  154.06    .045       0     189     .12       0
  274.36    .016       0
#XS Ineff= 2 , 0
                          219.02         2447.35
Permanent Ineff=
       F       F
Bank Sta=154.06,189
XS Rating Curve= 0 ,0
Exp/Cntr=0.3,0.1

Type RM Length L Ch R = 1 ,13830.2 ,253.1,206.2,144.5
XS GIS Cut Line= 5
2035076.63274549339703.8372705692035159.14952098339699.428441096
2035349.55106622339618.0699839472035400.26679365339577.683468896
2035434.18320635339548.804236455
#Sta/Elev= 30
       0 2484.52    30.5 2469.23    40.3 2465.22    50.2 2462.54    73.2 2460.12
    97.4 2459.06   108.1  2453.1   118.8 2452.04     133 2446.77   143.7  2444.6
   179.4 2443.91   190.1 2442.84     208 2444.21   211.5 2443.62   216.9 2441.32
   229.3 2440.28   243.6 2440.36   247.2  2441.4   254.3    2446   257.9 2446.28
   279.3 2446.28   294.1 2445.29   311.1 2449.96   315.1 2449.46   323.6 2445.69
   330.7 2445.04   336.1 2446.97   341.2 2449.86  379.982451.364   399.1 2452.27
#Mann= 4 ,-1 , 0
       0     .12       0   216.9    .045       0   247.2     .12       0
  379.98    .016       0
#XS Ineff= 2 , 0
                           309.6          2450.3
Permanent Ineff=
       F       F
Bank Sta=216.9,247.2
XS Rating Curve= 0 ,0
Exp/Cntr=0.3,0.1

Type RM Length L Ch R = 1 ,13624   ,47.2,122.9,193.5
XS GIS Cut Line= 2
2035367.31097781339836.9178221182035441.55884578339566.655582693
#Sta/Elev= 30
       0 2448.01    28.9 2448.19    61.8 2447.59    62.9  2447.5    66.3  2446.5
    69.8 2445.08    73.1  2444.3    76.5 2443.78    80.62442.146    83.3  2440.7
    86.7 2440.24    90.1 2440.35   107.1 2442.06   113.9 2443.06   120.7 2445.19
   124.1  2445.3   137.7 2444.91   144.7 2444.33     148 2443.85   151.4 2443.81
     165 2444.83   178.6 2445.06   195.6 2444.06     222 2444.41   236.4 2444.99
   239.8 2445.37     250 2448.56   260.2 2450.69   270.4 2452.01   280.3 2452.27
#Mann= 3 , 0 , 0
       0     .12       0    80.6    .045       0   107.1     .12       0
Bank Sta=80.6,107.1
XS Rating Curve= 0 ,0
Exp/Cntr=0.3,0.1

Type RM Length L Ch R = 1 ,13501.1 ,189.1,164.8,134.8
XS GIS Cut Line= 4
2035375.07346551339849.285366412 2035452.9392485339776.014735452
 2035639.7925893  339772.44903012035667.23232274339770.578314716
#Sta/Elev= 30
       0 2446.87       6 2446.65    15.6 2447.82    19.4 2447.93    34.7 2447.18
      42 2447.33    76.6 2446.19   105.8 2446.03   128.6 2444.22   134.3 2443.55
   138.32441.681   141.6 2440.35     158 2440.04   164.6 2440.17   167.9 2440.62
   171.2 2441.68   174.5 2442.93   177.7 2443.62   184.3 2444.14   187.6 2445.32
   194.1 2450.33   206.1 2458.57   220.4 2465.52   233.5 2473.53   239.6 2476.83
   246.6 2480.11     276 2492.09     3022503.755   315.6 2509.99   321.3  2511.4
#Mann= 6 ,-1 , 0
       0     .12       0    76.6     .08       0   128.6    .016       0
   138.3    .045       0   171.2    .016       0     302     .12       0
Bank Sta=138.3,171.2
XS Rating Curve= 0 ,0
Exp/Cntr=0.3,0.1

Type RM Length L Ch R = 1 ,13336.3 ,287.2,293.5,299.1
XS GIS Cut Line= 4
     2035352.535      340049.889      2035466.73      339974.685
     2035568.802       339905.31     2035687.303      339838.116
#Sta/Elev= 30
       0 2461.49     8.5 2462.13    32.1 2460.47    47.9 2460.24    85.9 2458.08
   105.6    2456   143.5  2453.1   160.3  2450.6  174.032447.804   193.1 2443.31
   200.2 2439.69   201.7 2439.14   205.7 2438.96   221.4  2439.4   232.9 2439.11
   235.6 2439.79   241.4  2442.7   245.3 2444.07   261.6 2444.98   264.9 2446.39
   268.8 2449.48   272.5 2451.36   291.3 2456.45   307.3 2462.05   321.8 2470.15
   332.8 2477.59     341 2482.11   359.2 2491.62   385.6 2504.19   396.4 2510.47
#Mann= 4 ,-1 , 0
       0     .12       0  174.03    .016       0   200.2    .045       0
   235.6     .12       0
Bank Sta=200.2,235.6
XS Rating Curve= 0 ,0
Exp/Cntr=0.3,0.1

Type RM Length L Ch R = 1 ,13042.8 ,290.1,278.6,265.6
XS GIS Cut Line= 4
     2035568.305      340239.945     2035652.538      340193.613
     2035769.878      340132.619     2035867.164      340086.806
#Sta/Elev= 30
       0 2454.75    20.3 2453.03    50.1 2451.81   87.832453.009    98.4 2451.96
   102.6 2450.82   111.8  2446.7  121.222441.411   124.8 2440.06   132.2 2438.29
   135.9 2436.95   139.6  2436.4   154.2 2436.25   181.2 2436.46     186 2437.09
   193.3 2439.68   198.2 2440.96   209.8 2441.67   220.9 2441.44   234.8 2443.24
   260.9  2451.2   268.2 2452.92   276.7 2453.94     289  2454.3   293.6 2454.83
   297.2 2455.83   311.7 2461.27   322.6 2467.08   333.5 2471.16   335.9 2472.75
#Mann= 5 ,-1 , 0
       0     .12       0   87.83    .016       0  121.22     .12       0
   135.9    .045       0     186     .12       0
Bank Sta=135.9,186
XS Rating Curve= 0 ,0
Exp/Cntr=0.3,0.1

Type RM Length L Ch R = 1 ,12764.2 ,353.8,387.2,421.5
XS GIS Cut Line= 4
      2035667.94      340474.362     2035836.729      340416.804
     2035896.612       340366.49     2036073.444      340201.943
#Sta/Elev= 30
       0 2447.28   15.392448.289    58.7 2447.29    97.2 2447.64   135.4 2446.82
  163.282447.045     170 2446.81     177 2445.94   189.6 2443.48   198.32441.115
   210.9 2437.09   223.92436.021   238.5 2435.05   245.5 2436.22   252.5 2438.97
   264.1 2440.34   289.8 2440.62     309 2439.19   316.4  2439.3   328.3 2441.69
   338.4 2445.92   342.8 2446.66   356.7 2447.13   383.6 2446.09   395.7  2446.8
   410.5 2448.61   434.3 2452.48   458.3 2455.02   468.4  2457.9   498.1 2461.05
#Mann= 6 ,-1 , 0
       0     .07       0   15.39     .12       0  163.28    .016       0
   198.3     .12       0   223.9    .045       0   245.5     .12       0
#XS Ineff= 2 , 0
                          283.98         2440.88
Permanent Ineff=
       F       F
Bank Sta=223.9,245.5
XS Rating Curve= 0 ,0
Exp/Cntr=0.3,0.1

Type RM Length L Ch R = 1 ,12377   ,735.3,779,735.6
XS GIS Cut Line= 5
     2035522.939      340713.818     2035872.241      340672.717
     2035981.397       340680.42     2036179.417      340664.131
      2036330.01      340644.993
#Sta/Elev= 30
       0 2445.88    40.5 2442.79  123.162439.183     133 2440.09   185.8 2438.68
  242.12 2439.52   294.8 2437.28   344.4 2439.31   377.3 2437.58   387.2 2432.25
   390.4 2431.55     397 2432.42   406.9 2437.81  449.872436.779  509.14 2436.12
   518.8 2436.68   531.9 2433.15   545.1 2432.94   561.6 2430.61   571.4 2429.81
   593.6 2430.98   610.9 2438.33   620.8 2440.47   630.7 2440.15   637.3  2441.4
   670.2 2461.38   688.5 2471.23   700.2 2475.86   769.5 2492.78   811.6 2497.77
#Mann= 7 ,-1 , 0
       0     .12       0  123.16     .07       0  242.12     .12       0
  449.87    .016       0  509.14     .12       0   561.6    .045       0
   593.6     .12       0
#XS Ineff= 2 , 0
          414.36 2437.59
Permanent Ineff=
       F       F
Bank Sta=561.6,593.6
XS Rating Curve= 0 ,0
Exp/Cntr=0.3,0.1

Type RM Length L Ch R = 1 ,11598   ,256.8,268.8,279.6
XS GIS Cut Line= 4
     2035542.702      341114.225     2035909.962      341005.581
     2036032.506      340964.629     2036311.785      340870.944
#Sta/Elev= 30
       0 2553.24    23.8 2541.26    89.9 2513.97   137.4 2491.82     165 2476.99
   192.4 2460.21   219.7 2440.68   240.3 2440.57   256.2    2437   291.6 2434.69
   322.2 2430.98   339.5 2434.73     384 2433.86   411.6 2435.15   418.6 2433.21
   425.5  2429.2   432.4 2427.26   453.1  2428.9   463.5 2430.22   484.3 2435.63
   515.2 2435.58     554 2441.07   644.7 2442.42     694 2441.15   716.1 2442.64
   736.9 2449.39   750.7 2458.65   761.1 2462.24   799.2 2487.46   806.8 2491.29
#Mann= 3 ,-1 , 0
       0     .12       0   425.5    .045       0   453.1     .12       0
Bank Sta=425.5,453.1
XS Rating Curve= 0 ,0
Exp/Cntr=0.3,0.1

Type RM Length L Ch R = 1 ,11329.2 ,330,319.4,303.9
XS GIS Cut Line= 4
     2035680.412        341265.7     2035942.772      341254.899
     2036039.184      341245.094     2036340.129      341166.224
#Sta/Elev= 30
       0 2516.85    17.2 2508.62    59.9 2484.02   132.2 2449.33     142 2440.99
   145.3 2439.94     165 2440.09   178.1 2434.75   233.9 2431.72   289.9 2432.37
   296.5 2431.27   299.8 2428.92   306.4 2426.65   327.2 2429.09   336.1 2433.06
   342.6 2434.08   420.2 2429.81   433.7  2432.6   468.6 2433.23     485 2432.46
   501.6 2429.77   519.6 2430.32     525 2431.59   535.5 2438.91   543.8 2441.72
   555.8  2443.3   576.4 2442.82   603.3 2444.85   640.6 2455.27   670.6 2461.16
#Mann= 3 ,-1 , 0
       0     .12       0   299.8    .045       0   327.2     .12       0
Bank Sta=299.8,327.2
XS Rating Curve= 0 ,0
Exp/Cntr=0.3,0.1

Type RM Length L Ch R = 1 ,11009.7 ,237.5,206.3,164.8
XS GIS Cut Line= 4
     2035720.871        341617.9     2035958.026      341530.981
     2036016.289      341516.973     2036322.204      341388.425
#Sta/Elev= 30
       0 2496.11    12.7 2491.75    59.1 2473.17    88.9 2464.26   105.5 2460.73
     115 2457.83   127.1  2452.7     136 2450.27   187.3 2443.05   202.4  2437.8
   223.1 2437.79   233.8  2434.1   253.9 2430.74   268.2 2430.55   273.9  2427.9
   281.1 2426.38   295.2 2426.75   299.92428.314   305.3 2430.71   312.1 2431.86
   386.3 2430.48   418.8 2431.26   441.4 2433.52   476.5 2438.52   514.9 2438.76
   556.7 2440.53   574.2 2438.29   604.3 2436.73   621.7 2438.58   644.3  2443.2
#Mann= 3 ,-1 , 0
       0     .12       0   273.9    .045       0   299.9     .12       0
Bank Sta=273.9,299.9
XS Rating Curve= 0 ,0
Exp/Cntr=0.3,0.1

Type RM Length L Ch R = 1 ,10803.4 ,131,333.4,404.1
XS GIS Cut Line= 4
     2035881.727      341787.811     2036080.204      341709.674
     2036124.768      341624.8222036446.69146494341376.129895451
#Sta/Elev= 30
       0  2493.8    10.2  2488.1    20.8 2486.35    31.3 2479.98    87.7 2451.47
   101.8 2445.66   108.9 2439.37   112.4 2437.48   131.6 2437.84   147.7 2434.16
   182.9 2432.44   230.2 2433.75   234.4 2432.78   240.4 2428.62   246.6 2426.98
   262.6  2427.1   268.4  2428.8   273.7 2430.92   285.4  2431.8   299.7 2431.19
   349.8 2432.61   453.4 2431.72   490.8 2432.78   555.3 2431.17   569.5 2431.52
   585.7 2433.28   627.6 2434.52   641.9 2437.81   702.2 2466.59   715.9 2471.36
#Mann= 3 ,-1 , 0
       0     .12       0   240.4    .045       0   268.4     .12       0
#XS Ineff= 2 , 0
                             500            2450
Permanent Ineff=
       F       F
Bank Sta=240.4,268.4
XS Rating Curve= 0 ,0
Exp/Cntr=0.3,0.1

Type RM Length L Ch R = 1 ,10470.1 ,99.9,226,222.1
XS GIS Cut Line= 4
     2035904.675      341794.576     2036331.097      341715.397
     2036415.045      341734.477     2036438.894      341739.246
#Sta/Elev= 30
       0 2482.33    19.7 2471.11    29.7 2466.54      53  2454.1    66.4 2448.25
    69.7 2445.61    76.4 2436.34    79.7 2435.38    86.4  2437.3    97.2 2437.65
   106.4 2436.93   116.4 2434.57   126.4 2433.88   169.1  2434.3   186.5 2433.36
   223.2 2433.27   253.2 2434.24   279.9 2431.87     352 2431.31   380.1 2431.84
   416.8 2431.09   440.2 2432.28   450.3 2431.15   462.12426.605   477.1 2425.66
   483.9  2426.7   487.3  2428.8   500.7 2439.59   510.1 2445.24   544.1 2460.59
#Mann= 3 ,-1 , 0
       0     .12       0   462.1    .045       0   483.9     .12       0
Bank Sta=462.1,483.9
XS Rating Curve= 0 ,0
Exp/Cntr=0.3,0.1

Type RM Length L Ch R = 1 ,10244   ,192.5,171.7,146.9
XS GIS Cut Line= 4
      2035891.32      341835.597     2036161.291      341821.287
     2036234.746      341835.597     2036410.826      341856.548
#Sta/Elev= 30
       0 2483.76     6.4 2479.49    19.6 2474.32    42.6 2461.06      53 2457.25
    62.3 2451.12    72.2  2442.6    75.4 2441.15    95.2 2439.82   108.3 2435.39
   134.6 2433.22   157.6 2434.91   164.1 2434.11   216.7 2434.71   239.7 2433.49
   282.6 2435.65  294.78 2426.85   302.1 2425.73   316.1 2425.87   321.7 2427.26
   329.4 2430.25   336.1 2431.35   369.3    2432   385.8 2430.98   427.6 2430.99
   441.4 2433.18   455.2 2436.65   468.8 2442.68   483.8 2447.61   522.5 2453.56
#Mann= 3 ,-1 , 0
       0     .12       0  294.78    .045       0   321.7     .12       0
#XS Ineff= 2 , 0
          279.48 2435.39
Permanent Ineff=
       F       F
Bank Sta=294.78,321.7
XS Rating Curve= 0 ,0
Exp/Cntr=0.3,0.1

Type RM Length L Ch R = 1 ,10072.3 ,338.2,336.9,281.5
XS GIS Cut Line= 4
     2035853.074      342036.712     2036219.703      341980.077
     2036282.444      341958.658     2036406.151      341939.159
#Sta/Elev= 30
       0 2450.61    45.2  2441.2    65.1 2438.82    78.4 2436.36      88  2432.7
    98.3 2434.14   122.5  2432.9   131.1 2430.01     136 2429.96   144.8 2429.65
   154.8 2430.31   181.3  2429.1   221.2 2428.55   237.8 2429.34   251.9 2430.87
   304.2 2431.47   323.8 2433.01   377.7 2432.05   384.4 2430.83   392.92426.695
   398.3 2425.59   411.3 2425.68   415.6 2426.74   422.5 2429.93   432.9 2429.93
   436.4 2430.82   449.7 2437.27   506.2 2452.73   519.5 2455.94   562.5 2462.61
#Mann= 5 ,-1 , 0
       0     .12       0   122.5    .016       0     136     .12       0
   392.9    .045       0   415.6     .12       0
Bank Sta=392.9,415.6
XS Rating Curve= 0 ,0
Exp/Cntr=0.3,0.1

Type RM Length L Ch R = 1 ,9735.4  ,348.4,276.4,237.3
XS GIS Cut Line= 3
     2035931.386      342243.892     2036133.626      342179.977
     2036422.422      342092.069
#Sta/Elev= 30
       0 2442.39    23.2    2437    33.5 2431.59    40.4  2430.7    43.9 2430.56
    50.8 2431.48      68 2431.22    81.7 2431.87    91.2 2431.35    98.9 2432.47
   118.8 2432.22   126.4 2432.42   133.3 2429.93   140.2 2426.29   143.7 2425.57
   164.8 2425.53   171.2 2426.22   178.1 2429.48   182.7 2430.46   226.2 2431.47
   267.3  2433.2   380.5 2433.84   390.8 2432.99   407.9 2433.66   442.2 2432.08
   466.2 2431.85     477 2432.68   486.8 2434.52   507.4  2440.2     514 2442.48
#Mann= 5 ,-1 , 0
       0     .12       0    98.9    .016       0   118.8     .12       0
   140.2    .045       0   171.2     .12       0
#XS Ineff= 2 , 0
              93    2440
Permanent Ineff=
       F       F
Bank Sta=140.2,171.2
XS Rating Curve= 0 ,0
Exp/Cntr=0.3,0.1

Type RM Length L Ch R = 1 ,9459    ,190.1,263.4,296.8
XS GIS Cut Line= 4
     2036264.729       342336.71     2036347.314      342272.511
     2036341.643      342174.692     2036452.811      342108.512
#Sta/Elev= 30
       0 2448.29    10.7 2448.24    50.4 2445.47    71.3 2442.86   104.2 2436.17
   123.8 2434.33   130.4  2433.2     137 2431.58   146.9 2430.27   153.4  2428.5
   156.7 2426.18     160 2424.24   166.6 2424.04   176.4 2424.12   179.7 2424.89
  181.832426.387   186.3 2429.14   192.9 2429.45   202.6 2431.81   216.7 2431.48
   241.3 2432.24   254.9 2431.96   277.8 2429.98   285.7 2430.02   290.5 2430.43
   299.1 2432.15   305.5 2434.32   319.8 2441.34   327.5 2444.48     332 2446.87
#Mann= 3 ,-1 , 0
       0     .12       0   156.7    .045       0  181.83     .12       0
Bank Sta=156.7,181.83
XS Rating Curve= 0 ,0
Exp/Cntr=0.3,0.1

Type RM Length L Ch R = 1 ,9195.6  ,306.6,322.2,336.9
XS GIS Cut Line= 3
     2036320.603       342356.46     2036506.626      342298.268
     2036641.134       342264.88
#Sta/Elev= 30
       0 2446.84     6.7 2446.39    27.7 2443.67    65.7 2435.96    79.5 2434.21
    98.3 2433.15   113.8 2432.98   121.9 2431.83   127.6 2431.64   132.4  2432.1
   137.9 2434.12   141.3 2434.85   148.4 2433.94   175.7 2432.02   199.7 2431.28
   209.8 2431.67   213.2 2430.89     225 2426.25   230.1 2424.69   233.5 2424.23
   250.4 2424.36   256.22426.311   267.3 2428.15   270.7 2430.07   280.8 2438.63
     291 2446.15   304.5 2456.98   314.6 2463.39   327.9 2473.12   333.5 2476.21
#Mann= 3 ,-1 , 0
       0     .12       0     225    .045       0   256.2     .12       0
#XS Ineff= 2 , 0
          141.07    2435
Permanent Ineff=
       F       F
Bank Sta=225,256.2
XS Rating Curve= 0 ,0
Exp/Cntr=0.3,0.1

Type RM Length L Ch R = 1 ,8873.3  ,284.5,289.6,294.9
XS GIS Cut Line= 4
2036345.66972489342592.719042641     2036443.664      342597.812
     2036536.708      342601.258     2036622.196       342605.31
#Sta/Elev= 30
       0 2449.97   12.762448.732    24.6  2447.9   37.982445.585   42.332443.997
    47.6 2441.83    71.92441.766    80.4 2441.22    90.3 2438.98   103.4 2432.24
   106.7 2431.39   116.5 2431.68   119.8 2430.65   126.4 2426.51   129.7 2424.83
     133 2424.21   151.4  2424.1   155.9 2424.14   159.2 2424.89   162.5 2426.77
   165.8 2428.04   182.2 2429.47     192 2432.42   205.2  2433.8   208.5 2434.96
   234.7  2448.2   247.9 2453.98   261.2  2462.4   274.2 2467.21   276.8 2468.61
#Mann= 7 ,-1 , 0
       0     .12       0   12.76    .016       0   37.98     .12       0
   42.33    .016       0    71.9     .12       0   126.4    .045       0
   162.5     .12       0
Bank Sta=126.4,162.5
XS Rating Curve= 0 ,0
Exp/Cntr=0.3,0.1

Type RM Length L Ch R = 1 ,8583.8  ,384.5,373.2,361.2
XS GIS Cut Line= 4
 2036304.1565777342870.345957359     2036465.605      342872.554
     2036548.585      342885.553     2036642.917      342892.752
#Sta/Elev= 30
       0 2453.51    33.2 2441.83    43.1 2440.47   54.122440.839    69.3 2441.09
   83.682438.925    92.3 2437.25   108.7 2432.69   151.4  2433.4   157.9 2432.26
   164.5 2429.53   167.8 2428.89   174.5 2428.19   184.4 2428.08   187.8  2427.5
   191.7 2426.07   194.4 2425.13   197.7 2424.81   217.7 2424.32   222.2 2426.01
   233.7 2432.43   242.3 2436.06   250.2 2438.65   260.7  2440.9   267.3 2441.28
   273.8 2442.35   306.7 2451.52   316.6  2453.1   323.2 2455.42   340.1 2460.05
#Mann= 5 ,-1 , 0
       0     .12       0   54.12    .016       0   83.68     .12       0
   191.7    .045       0   222.2     .12       0
#XS Ineff= 2 , 0
          142.12 2433.68
Permanent Ineff=
       F       F
Bank Sta=191.7,222.2
XS Rating Curve= 0 ,0
Exp/Cntr=0.3,0.1

Type RM Length L Ch R = 1 ,8210.6  ,346.7,283,218.7
XS GIS Cut Line= 3
     2036232.116      343253.178     2036496.007      343229.865
2036642.70505085343126.420100445
#Sta/Elev= 30
       0 2497.66    13.5  2493.2      53 2474.67      76 2465.27   105.7 2453.83
   125.4 2446.99   128.7 2444.02     132  2439.6   135.3    2436   138.6 2434.19
  152.122434.572   155.1 2434.49   158.4  2433.4     165  2427.2   167.4 2425.82
     172 2424.42   187.2 2424.16   191.3 2424.69   194.6 2426.21   201.2 2429.32
   214.3 2431.96   227.5 2433.91   247.7 2441.04   253.8 2442.66   257.2  2443.1
   298.6 2445.27   314.2 2445.46   351.8  2448.6     396 2451.05   444.4 2454.61
#Mann= 4 ,-1 , 0
       0     .12       0  152.12    .016       0   167.4    .045       0
   194.6     .12       0
Bank Sta=167.4,194.6
XS Rating Curve= 0 ,0
Exp/Cntr=0.3,0.1

Type RM Length L Ch R = 1 ,7927.7  ,262.3,253.8,245.5
XS GIS Cut Line= 4
     2036383.494       343633.67     2036563.789      343514.443
     2036595.776      343399.578     2036690.286      343155.308
#Sta/Elev= 30
       0 2530.35    19.5 2522.17      52 2511.19    63.2 2508.15    75.8 2503.14
   117.8 2484.92   131.8 2477.79   155.5 2467.27   206.6 2451.83     210 2449.48
  218.962441.056   224.3 2436.49   227.7 2435.61   237.9 2437.27   251.6 2436.13
  264.16 2424.33   268.6 2422.79   283.8 2422.73     289 2422.81   293.3 2424.48
   302.4 2429.61   306.1 2430.74   329.1 2430.15   344.6 2431.24     408 2442.17
   428.3  2442.3   463.8 2446.61   498.6 2448.45   544.3 2452.23   597.3 2454.26
#Mann= 4 ,-1 , 0
       0     .12       0  218.96    .016       0  264.16    .045       0
   293.3     .12       0
Bank Sta=264.16,293.3
XS Rating Curve= 0 ,0
Exp/Cntr=0.3,0.1

Type RM Length L Ch R = 1 ,7673.8  ,391.6,435,474.6
XS GIS Cut Line= 3
     2036674.292       343720.91     2036821.145      343563.879
     2036853.132      343289.075
#Sta/Elev= 30
       0 2451.72    6.912447.126    11.1 2445.45      27 2445.17   50.152442.593
    73.5  2438.3   101.3 2437.07   131.2 2434.78     160 2434.62   174.4 2433.17
   190.1 2434.28   203.6 2434.22   219.8 2432.96   229.7  2434.5   239.7 2433.63
   259.5 2433.47   266.1 2432.36   279.3 2425.62     289 2423.48   295.8 2422.68
   322.2 2422.83   330.4 2423.58     352 2427.87   381.7 2427.98   414.7 2431.47
   421.3 2433.93   447.7 2446.52     451  2447.5   461.4 2449.69   491.7 2453.43
#Mann= 5 ,-1 , 0
       0     .12       0    6.91    .016       0   50.15     .12       0
     289    .045       0   330.4     .12       0
Bank Sta=289,330.4
XS Rating Curve= 0 ,0
Exp/Cntr=0.3,0.1

Type RM Length L Ch R = 1 ,7238.8  ,455.4,448,442.9
XS GIS Cut Line= 4
     2036796.427      343888.118     2036995.623      343824.143
     2037071.231      343761.621     2037183.188      343665.658
#Sta/Elev= 30
       0  2448.2     .772447.684     7.2 2443.06    10.6 2441.34    19.2 2440.45
    31.3  2437.8    37.5 2437.17      52 2438.26   124.3 2432.74   167.9 2431.71
   196.3 2432.16   223.6 2431.06   230.6 2429.29   239.9 2421.92   244.8 2419.59
   254.5    2419   275.1 2419.16   279.5  2420.1   283.2 2422.08   287.4 2423.67
   291.7 2424.14   305.1  2424.8   316.1 2424.52   330.3 2426.01   356.3  2425.9
   369.2 2427.41   382.2 2427.69   393.6 2430.82   421.1 2436.43   454.8 2447.46
#Mann= 4 ,-1 , 0
       0    .016       0     .77     .12       0   239.9    .045       0
   283.2     .12       0
Bank Sta=239.9,283.2
XS Rating Curve= 0 ,0
Exp/Cntr=0.3,0.1

Type RM Length L Ch R = 1 ,6790.8  ,517.3,530,542.6
XS GIS Cut Line= 4
      2037172.66      344240.758     2037366.391      344068.413
     2037476.631      343962.665     2037558.598      343889.208
#Sta/Elev= 30
       0 2455.47   11.352454.655    58.5 2450.14    76.4 2449.46   128.2 2445.68
   151.5  2443.6   164.3 2441.72     195 2440.72   209.6 2438.66   260.9 2434.27
   274.6 2432.28   284.2 2429.79   288.9 2428.16   307.1 2420.05   310.9 2418.95
   329.1 2418.73   342.8    2419   347.3 2420.03   351.2 2421.85   356.4 2423.21
   379.1 2424.35   402.7 2431.26     411  2434.4   451.5 2451.67   468.3 2459.68
   494.7 2475.66   507.9 2484.93   511.4 2486.42   518.4    2488   522.1 2490.24
#Mann= 4 ,-1 , 0
       0    .016       0   11.35     .12       0   307.1    .045       0
   347.3     .12       0
Bank Sta=307.1,347.3
XS Rating Curve= 0 ,0
Exp/Cntr=0.3,0.1

Type RM Length L Ch R = 1 ,6260.8  ,320.8,352.3,383.2
XS GIS Cut Line= 4
     2037233.378      344569.319     2037614.674      344497.323
     2037774.261      344401.125     2037849.223      344358.663
#Sta/Elev= 30
       0 2455.91    29.7 2438.85   37.012432.528    43.1 2427.81    46.4 2426.85
    53.1 2428.28   67.072428.379   103.2  2423.3   176.6 2421.71   206.7 2419.87
  247.422419.823   409.8 2423.95   421.3 2420.15   432.4 2418.41   436.6 2416.06
     443 2414.74   466.1 2415.28  469.09 2416.42   474.9 2419.96   482.8 2421.07
   495.9 2421.04   509.4 2422.67   537.8 2422.25   547.7 2423.65   555.4 2427.99
   574.5 2443.16   586.4 2450.71     629 2486.88     641 2493.56   660.5 2501.23
#Mann= 6 ,-1 , 0
       0     .12       0   37.01    .016       0   67.07     .08       0
  247.42     .12       0   436.6    .045       0  469.09     .12       0
#XS Ineff= 2 , 0
          406.78 2424.12
Permanent Ineff=
       F       F
Bank Sta=436.6,469.09
XS Rating Curve= 0 ,0
Exp/Cntr=0.3,0.1

Type RM Length L Ch R = 1 ,5908.5  ,632.8,607.6,578
XS GIS Cut Line= 4
      2037233.95       344689.48     2037785.032      344736.799
     2037921.432      344742.908     2038115.744      344747.178
#Sta/Elev= 30
       0 2454.79    27.8 2439.84   35.932432.082   43.952425.735    48.5 2423.52
   65.572424.948   95.222420.991   196.7 2417.01     325  2421.7   387.7  2420.4
   466.7 2421.79   499.6 2420.43   529.3 2424.71     549 2422.62   581.9  2422.8
   598.3 2419.57   608.1 2419.13   617.5  2415.5   627.9 2414.34  648.06 2415.73
   665.6 2432.02   687.6 2442.31   713.2  2447.2     746 2442.23   759.2 2443.97
   777.5 2455.65     792 2469.52   801.8 2476.01     844 2490.85     884  2498.5
#Mann= 7 ,-1 , 0
       0     .12       0   35.93    .016       0   43.95     .12       0
   65.57    .016       0   95.22     .12       0   617.5    .045       0
  648.06     .12       0
#XS Ineff= 2 , 0
          526.29 2424.87
Permanent Ineff=
       F       F
Bank Sta=617.5,648.06
XS Rating Curve= 0 ,0
Exp/Cntr=0.3,0.1

Type RM Length L Ch R = 1 ,5300.9  ,275.8,275.6,273.7
XS GIS Cut Line= 4
     2037407.493      345099.559     2037456.538      345074.268
     2037620.152      345004.083     2037710.666       345013.41
#Sta/Elev= 30
       0 2494.99     6.8 2494.34    10.5    2493      40  2471.1    43.7 2468.09
    49.6  2462.1    59.5 2454.36    65.5 2447.92    72.6  2439.5    76.92435.874
    79.8 2434.56    83.3 2433.76    97.6 2432.86   101.2 2431.26  109.04  2423.1
   115.5 2416.89   119.4 2414.64   124.4 2412.99   129.4  2412.5     144 2412.67
   149.3 2414.92   154.7 2417.62   161.9 2419.12   196.9 2418.73   211.9 2419.34
   226.9  2421.6  237.272424.911   249.7 2427.88   266.2 2430.17   324.2 2433.52
#Mann= 6 ,-1 , 0
       0     .12       0    76.9    .016       0  109.04     .12       0
   119.4    .045       0   149.3     .07       0  237.27     .06       0
#XS Ineff= 2 , 0
                          176.29         2419.72
Permanent Ineff=
       F       F
Bank Sta=119.4,149.3
XS Rating Curve= 0 ,0
Exp/Cntr=0.5,0.3

Type RM Length L Ch R = 1 ,5025.3  ,182.3,182.3,182.3
XS GIS Cut Line= 3
      2037512.44       345324.82     2037789.646      345205.984
     2038033.862      345111.504
#Sta/Elev= 30
       0 2483.03    10.2 2481.66    13.7 2480.38    31.6 2468.49    67.3 2448.08
    92.3 2436.89  103.632432.779   113.7 2425.85   135.1  2425.9  153.71 2423.11
   163.6 2420.03   172.5 2419.85     185 2417.79     200  2416.6   202.9 2415.97
   207.5 2413.19     210 2411.65   227.5 2411.32   238.6 2411.65   242.5 2413.34
   249.3 2419.43     260  2427.3   263.6 2429.01   277.4 2432.94  282.26 2433.34
   297.7 2433.62   348.6 2437.54   457.2    2447   495.2 2451.16   563.5 2456.56
#Mann= 6 ,-1 , 0
       0     .12       0  103.63    .016       0  153.71     .12       0
   207.5    .045       0   242.5     .12       0  282.26     .06       0
Bank Sta=207.5,242.5
XS Rating Curve= 0 ,0
Exp/Cntr=0.5,0.3

Type RM Length L Ch R = 1 ,4843    ,46.2,46.2,46.2
XS GIS Cut Line= 4
2037516.64794226345428.5701620842037682.52770469345398.886415123
2037796.02438425345449.5233952332037988.09568811345351.741640538
#Sta/Elev= 30
       0 2493.23    15.2 2485.91    28.5 2481.44    38.5 2480.94    45.2 2478.64
    61.9 2465.55    95.2 2445.24   105.2 2437.73   121.9 2435.67   128.5 2431.43
   138.5  2427.5   151.9 2419.84   190.1 2418.61   197.3 2415.89   204.4 2412.11
   211.6 2410.68   218.8 2411.28   229.6 2415.36   236.8  2417.3   276.3 2416.33
   290.7  2418.5   301.6 2422.28   301.6 2422.31   321.1 2426.77     348 2430.11
   384.6  2431.1   417.3 2434.93   465.1 2438.24   485.7 2437.56   508.3 2431.66
#Mann= 6 ,-1 , 0
       0     .12       0   197.3    .045       0   229.6     .12       0
   301.6    .016       0   384.6     .12       0   465.1     .08       0
#XS Ineff= 2 , 0
                          238.21         2416.39
Permanent Ineff=
       F       F
Bank Sta=197.3,229.6
XS Rating Curve= 0 ,0
Exp/Cntr(USF)=0,0
Exp/Cntr=0.5,0.3

Type RM Length L Ch R = 1 ,4797    ,97.1,97.1,97.1
XS GIS Cut Line= 4
2037504.42522292345477.4610394322037659.82836878345435.554573134
2037799.51658977345498.414272581 2037993.3339964345370.948770925
#Sta/Elev= 30
       0 2510.42    21.8 2497.32    31.6 2490.28    38.4 2488.12    48.5 2482.28
    58.9 2481.19    65.5  2478.6    79.1 2468.14   109.7 2448.35   116.5 2442.01
   136.9 2438.41   153.9 2429.22   175.1 2423.35   182.3 2422.89   196.6  2416.3
   209.3 2412.75   217.9 2410.18   236.2 2410.02   255.2 2413.71   262.6 2415.03
   331.8  2417.7   350.6 2421.97   362.6 2424.41   378.3 2425.19   404.4 2428.37
   465.9 2433.33   497.6 2436.16   529.8 2441.32   539.3 2441.74   546.1 2441.38
#Mann= 7 ,-1 , 0
       0     .12       0   209.3    .045       0   255.2     .12       0
   350.6    .016       0   404.4     .12       0   465.9     .08       0
   539.3     .12       0
#XS Ineff= 2 , 0
                          272.38          2415.8
Permanent Ineff=
       F       F
Bank Sta=209.3,255.2
XS Rating Curve= 0 ,0
Exp/Cntr(USF)=0,0
Exp/Cntr=0.5,0.3

Type RM Length L Ch R = 1 ,4699.7  ,561.2,538,529.5
XS GIS Cut Line= 5
     2037461.766      345770.422       2037685.4      345614.375
     2037812.064      345507.122     2037834.389      345490.517
     2037996.751      345385.521
#Sta/Elev= 30
       0 2547.73     9.2  2544.7    51.7 2523.99    64.4 2519.96   120.5 2496.99
   137.7 2487.33   165.7 2482.24   221.2 2461.19   233.2 2460.81     267 2451.91
   300.4 2435.82     309 2435.23   320.7 2440.37   333.4 2438.48   336.9 2436.54
   350.6 2422.34   367.8 2411.29   376.4 2410.03   399.8  2411.5   409.1 2412.03
   424.72415.856   455.8 2418.39   466.1 2420.87   484.1  2423.6  497.562423.229
   504.4 2425.96   531.5  2429.1  567.91 2431.25   621.7 2435.71   659.8 2442.77
#Mann= 7 ,-1 , 0
       0     .12       0   367.8    .045       0   399.8     .12       0
   424.7    .016       0   466.1     .12       0  497.56     .08       0
  567.91     .12       0
Bank Sta=367.8,399.8
XS Rating Curve= 0 ,0
Exp/Cntr=0.3,0.1

Type RM Length L Ch R = 1 ,4161.7  ,412.8,441.2,462.5
XS GIS Cut Line= 4
      2037852.34      346115.193     2037960.043      346055.957
     2038048.522      345944.601     2038226.532      345696.716
#Sta/Elev= 30
       0 2445.12    30.9  2442.6    42.1 2440.98    83.3 2428.21    97.5 2421.84
   109.3 2417.79   131.5 2421.03   140.9 2421.09     152  2418.3   156.7 2417.94
   168.4 2419.96   172.6 2419.55     186 2415.74   196.4 2407.23   198.7  2406.1
   209.5 2405.91   219.5 2406.08   222.8 2407.16   230.6 2409.91   248.8 2412.66
     290 2412.28  351.15 2413.12  387.522413.814   402.8 2413.26   412.2 2415.13
  423.882416.134  449.142417.463   495.8 2417.39  532.972420.855   570.3 2424.53
#Mann= 8 ,-1 , 0
       0     .12       0   196.4    .045       0   222.8     .12       0
  351.15     .08       0  387.52    .016       0  423.88     .08       0
  449.14     .12       0  532.97     .06       0
#XS Ineff= 2 , 0
                             270         2414.26
Permanent Ineff=
       F       F
Bank Sta=196.4,222.8
XS Rating Curve= 0 ,0
Exp/Cntr=0.5,0.3

Type RM Length L Ch R = 1 ,3720.5  ,214.6,262.4,315.3
XS GIS Cut Line= 4
     2037978.351      346234.132      2038284.48      346159.933
     2038376.081      346111.515     2038450.973      346075.321
#Sta/Elev= 30
       0 2440.11    23.1  2437.3    39.9 2432.91    53.5 2427.17    80.5 2413.61
    83.8 2412.95   131.1 2411.89  146.392410.334   164.9 2408.63     188 2412.67
   198.6 2413.37   242.4 2413.32  271.772410.892   286.4 2410.58   349.6 2412.11
   354.1 2410.48   360.5 2405.82   371.5 2404.64   383.6 2404.72   388.5 2406.05
   394.9 2410.18  403.362410.846   417.1 2412.47  436.442413.206     439 2414.64
   446.3 2421.92   454.4 2426.07   464.5 2429.71   493.5 2436.49   501.8 2439.47
#Mann= 7 ,-1 , 0
       0     .12       0  146.39     .06       0  271.77     .12       0
   360.5    .045       0   388.5     .12       0  403.36    .016       0
  436.44     .12       0
#XS Ineff= 2 , 0
          346.64 2412.27
Permanent Ineff=
       F       F
Bank Sta=360.5,388.5
XS Rating Curve= 0 ,0
Exp/Cntr=0.5,0.3

Type RM Length L Ch R = 1 ,3458.1  ,333.4,267.4,196.9
XS GIS Cut Line= 4
     2038002.838      346255.535     2038146.783      346290.867
     2038238.385      346340.593     2038439.908      346344.519
#Sta/Elev= 30
       0 2434.76       8 2431.42    28.4 2419.82    45.2  2412.8    68.8 2411.88
    97.9 2412.98   150.3 2413.25   153.8 2412.92   157.5 2411.43     165 2404.88
   167.2 2403.63   171.2 2402.54   181.7 2402.42     185 2402.71  187.96 2403.89
   191.1 2405.58   193.8 2406.07   209.8 2406.75  225.742409.366   257.6 2410.75
   277.3 2410.13     297 2411.63   317.62411.907   333.1  2412.1   342.9 2413.04
   364.3 2417.47   385.6 2421.01   405.3 2426.94   441.1 2439.88     454 2443.21
#Mann= 5 ,-1 , 0
       0     .12       0   167.2    .045       0  187.96     .12       0
  225.74    .016       0   317.6     .12       0
#XS Ineff= 2 , 0
                          259.31         2411.26
Permanent Ineff=
       F       F
Bank Sta=167.2,187.96
XS Rating Curve= 0 ,0
Exp/Cntr=0.3,0.1

Type RM Length L Ch R = 1 ,3190.7  ,288.6,296.2,302
XS GIS Cut Line= 3
     2038204.479      346582.759     2038297.259      346472.887
     2038417.604      346392.871
#Sta/Elev= 30
       0 2440.53       7 2439.03    12.9 2437.03      25 2432.49    30.1 2429.94
    36.2 2425.76    45.6 2415.47    50.1 2412.69    55.5 2411.52    67.1 2413.02
    71.1 2411.45    80.4 2406.08    87.7 2403.01      92 2401.68    97.1 2401.31
     110 2401.88     113  2403.2  114.832404.349   121.6 2408.75   127.2  2409.9
   136.3 2410.25     148 2409.47  157.172410.274   181.7 2411.33   201.4 2413.12
   243.7 2412.41   254.5 2412.76   259.2 2414.36   268.4 2420.66   288.3 2428.88
#Mann= 5 ,-1 , 0
       0     .12       0    87.7    .045       0     113     .12       0
  114.83    .016       0  157.17     .12       0
Bank Sta=87.7,113
XS Rating Curve= 0 ,0
Exp/Cntr=0.3,0.1

Type RM Length L Ch R = 1 ,2894.5  ,247.2,267.9,288.2
XS GIS Cut Line= 3
      2038400.94      346781.974     2038485.129      346707.526
     2038615.189      346593.915
#Sta/Elev= 30
       0 2426.65    19.5 2424.92    31.1 2422.74    46.3 2418.07    61.1 2412.52
    65.9 2410.17    68.3 2409.38      71 2408.82      79 2408.51    83.3 2407.54
    87.7 2405.87    95.8 2401.67   100.8 2401.09   110.7  2400.8   125.6 2400.98
   127.1 2401.46   128.7 2402.71   131.4 2405.55   133.4 2406.95   135.7 2408.09
  145.782407.241   160.5 2407.49   166.3 2408.23     175 2409.87     1852410.601
   196.8 2411.06   205.4 2415.12   221.7 2420.74   240.4 2425.81   285.1 2440.11
#Mann= 5 ,-1 , 0
       0     .12       0    95.8    .045       0   127.1     .12       0
  145.78    .016       0     185     .12       0
Bank Sta=95.8,127.1
XS Rating Curve= 0 ,0
Exp/Cntr=0.3,0.1

Type RM Length L Ch R = 1 ,2626.6  ,288.6,285,280.4
XS GIS Cut Line= 2
     2038506.646      346972.642     2038767.055      346882.349
#Sta/Elev= 30
       0 2416.18    27.1 2411.27    44.5 2409.81    72.3 2409.34    83.2 2406.96
    96.6  2406.3   103.5 2404.59   111.6 2403.21   117.4 2401.03   124.3 2399.51
   131.3 2399.47   138.2 2399.98   141.7 2401.05   145.2 2402.96   148.7  2404.3
   155.6 2405.29  160.15 2405.54     173  2405.8   176.4 2407.39   179.9 2410.74
   183.4  2413.6   186.8 2415.59  191.422417.327   198.5 2420.73   207.7 2424.08
   212.1 2425.33   222.4 2427.45   252.8 2431.86   259.8 2432.06   275.6 2433.86
#Mann= 5 ,-1 , 0
       0     .12       0   117.4    .045       0   141.7     .12       0
  160.15    .016       0  191.42     .12       0
Bank Sta=117.4,141.7
XS Rating Curve= 0 ,0
Exp/Cntr=0.5,0.3

Type RM Length L Ch R = 1 ,2341.6  ,294.6,270.6,246.9
XS GIS Cut Line= 2
     2038625.727       347234.36     2038895.297      347115.279
#Sta/Elev= 30
       0 2416.29    18.1 2413.16    41.3 2411.34    49.1 2408.67    52.1 2408.11
    55.6 2408.11    62.8 2408.88    66.4 2408.58    78.9 2403.73    86.4 2401.73
    91.2 2399.27    95.1 2397.85   102.3 2397.56   116.3 2397.67   118.8 2398.24
   121.3 2399.33   127.4 2403.39  132.112404.283   148.6  2404.9   164.42406.992
  196.692407.147  221.522407.239   235.7 2407.56   255.6 2407.25   260.6 2407.54
   269.8 2408.84   277.9 2412.54   285.5  2413.9   287.9 2414.66   294.7  2418.6
#Mann= 7 ,-1 , 0
       0     .12       0    91.2    .045       0   121.3     .12       0
  132.11    .016       0   164.4     .12       0  196.69     .08       0
  221.52     .12       0
Bank Sta=91.2,121.3
XS Rating Curve= 0 ,0
Exp/Cntr=0.3,0.1

Type RM Length L Ch R = 1 ,2071    ,117.5,117.5,117.5
XS GIS Cut Line= 2
2038726.28452496347579.4854944522039015.85121006347240.915216491
#Sta/Elev= 30
       0 2443.34    19.1 2435.29    33.2  2430.2    59.9 2422.09    82.1 2416.74
    93.7 2415.11     110 2409.37     124 2407.29   140.3 2406.34   189.2 2406.28
   196.2 2404.57   205.4 2399.14   209.1 2396.96   213.4 2396.12     222 2396.53
   228.7 2399.46     231 2400.86     235 2402.02   249.7 2401.64   256.7 2403.21
   261.8 2403.92   276.9 2403.97   282.4  2403.8   295.4 2405.62     317    2407
     380 2408.83   407.9 2410.44   416.3 2412.06   438.1 2418.96   445.5 2420.53
#Mann= 6 ,-1 , 0
       0     .06       0   140.3     .12       0   205.4    .045       0
   228.7     .06       0   256.7    .016       0   276.9     .06       0
#XS Ineff= 2 , 0
          184.85    2410
Permanent Ineff=
       F       F
Bank Sta=205.4,228.7
XS Rating Curve= 0 ,0
Exp/Cntr=0.5,0.3

Type RM Length L Ch R = 1 ,1953    ,41.6,41.6,41.6
XS GIS Cut Line= 4
2038863.35274633347632.9871838092038936.67229976347521.862235634
2038987.07949275347440.5233560432039077.58331652347284.719304994
#Sta/Elev= 30
       0 2423.72    22.5 2417.93    42.2 2413.97    51.7 2412.37    65.8 2411.16
    93.3 2406.67    97.2 2406.08   112.9 2405.25   131.6 2405.09   140.3 2404.46
   151.9 2401.22   153.6 2400.39   159.6 2396.33   171.2 2395.98   175.1 2396.09
   184.6 2400.66   187.5 2401.83   205.9 2403.93   217.5 2404.89   232.9 2405.42
   237.8 2405.14   246.7 2405.39   263.2 2408.16   270.7 2408.94   320.1 2409.28
   365.7 2410.55   373.9 2411.29   385.9 2414.39   399.8 2419.69     409 2422.67
#Mann= 6 ,-1 , 0
       0     .06       0    93.3     .12       0   153.6    .045       0
   184.6     .06       0   237.8    .016       0   320.1     .06       0
#XS Ineff= 2 , 0
          120.27 2404.23   225.5         2404.27
Permanent Ineff=
       F       F
Bank Sta=153.6,184.6
XS Rating Curve= 0 ,0
Exp/Cntr(USF)=0,0
Exp/Cntr=0.5,0.3

Type RM Length L Ch R = 1 ,1912    ,126.6,126.6,126.6
XS GIS Cut Line= 4
2038911.46870327347650.1714541452038969.89522241347547.065832128
2039011.13747122347480.6199868272039109.66062115 347306.48604742
#Sta/Elev= 30
       0 2423.19    11.2 2419.34    33.8 2412.88    67.8  2409.3    79.1 2407.63
    97.2  2405.1   128.3 2404.85   132.2 2403.62  135.54 2400.55   136.1 2399.78
   139.9 2397.29   143.8 2396.33   161.8 2395.85   166.9 2396.21   173.7 2400.49
   178.4 2401.77   190.4 2403.24   205.3 2406.19   209.1 2406.63   212.9 2406.22
   220.4 2405.45   231.7 2405.73   245.7  2405.1   267.3 2409.09     326 2409.92
   361.2 2411.01   363.7 2411.33   370.2 2413.56   390.1 2422.47   396.8 2424.56
#Mann= 6 ,-1 , 0
       0     .06       0    79.1     .12       0  135.54    .045       0
   173.7     .06       0   212.9    .016       0   267.3     .06       0
#XS Ineff= 2 , 0
          120.71 2404.31  202.67         2404.27
Permanent Ineff=
       F       F
Bank Sta=135.54,173.7
XS Rating Curve= 0 ,0
Exp/Cntr(USF)=0,0
Exp/Cntr=0.5,0.3
